--- SpringCrk2.prj (project) ---

Proj Title=SpringCrk2
Current Plan=p01
Default Exp/Contr=0,0
English Units
Geom File=g01
Flow File=f01
Plan File=p01
BEGIN DESCRIPTION:
AMEC Environment & Infrastructure, 2013
Projection: NAD 1983 State Plane West Virginia South FIPS 4702 (US Feet)
Vertical Datum: NAVD 1988
END DESCRIPTION:
DSS Export Rating Curves= 0
DSS Export Rating Curve Sorted= 0
DSS Export Volume Flow Curves= 0
DXF OffsetX= 0
DXF OffsetY= 0
DXF ScaleX= 0
DXF ScaleY= 0

--- SpringCrk2.p01 (plan) ---

Plan Title=Floodplain
Program Version=4.00
Geom File=g01
Flow File=f01
K Sum by GR=0
Std Step Tol=0.01
Critical Tol=0.01
Num of Std Step Trials=20
Max Error Tol=0.3
Flow Tol Ratio=0.001
Split Flow NTrial=30
Split Flow Tol=0.02
Split Flow Ratio=0.02
Log Output Level=0
Friction Slope Method=1
Unsteady Friction Slope Method=2
Unsteady Bridges Friction Slope Method=1
Global Log Level=0
CheckData=False
Run HTab=0
Run UNet=0
Run PostProcess=0
UNET Theta=0
UNET Theta Warmup=0
UNET ZTol=0
UNET ZSATol=0
UNET MxIter=0
UNET MaxInSteps=0
UNET DtIC=0
UNET DtMin=0
UNET MaxCRTS=0
UNET WFStab=0
UNET SFStab=0
UNET WFX=0
UNET SFX=0
UNET DSS MLevel=0
UNET DZMax Abort=0
UNET Convert EG Bridges=0
UNET Use Existing IB Tables=0
UNET Froude Limit=0
UNET Froude Power=0
Write IC File=0
Echo Input=False
Echo Output=False
Write Detailed=0

--- SpringCrk2.f01 (steady flow) ---

Flow Title=NFF Regression Equation
Program Version=4.10
Number of Profiles= 1
Profile Names=P100yr
River Rch & RM=SpringCrk2,Main            ,66291.3
7096.928
River Rch & RM=SpringCrk2,Main            ,62737.7
7161.471
River Rch & RM=SpringCrk2,Main            ,62339.6
 7328.63
River Rch & RM=SpringCrk2,Main            ,54459.4
7422.252
River Rch & RM=SpringCrk2,Main            ,53943.7
7620.523
River Rch & RM=SpringCrk2,Main            ,52476.2
7634.287
River Rch & RM=SpringCrk2,Main            ,51940.7
7667.061
River Rch & RM=SpringCrk2,Main            ,46963.5
7733.457
River Rch & RM=SpringCrk2,Main            ,46745.1
 7821.56
River Rch & RM=SpringCrk2,Main            ,37232.7
7897.737
River Rch & RM=SpringCrk2,Main            ,36397.5
8194.884
River Rch & RM=SpringCrk2,Main            ,19938.3
8411.332
River Rch & RM=SpringCrk2,Main            ,19558.7
9476.099
River Rch & RM=SpringCrk2,Main            ,9541.8
9718.641
River Rch & RM=SpringCrk2,Main            ,8733.5
9955.497
River Rch & RM=SpringCrk2,Main            ,85.6
 10209.9
Boundary for River Rch & Prof#=SpringCrk2,Main            , 1
Up Type= 0
Dn Type= 3
Dn Slope=0.0003
DSS Import GetInterval= 0
DSS Import GetPeak= 0
DSS Import FillOption= 0

--- SpringCrk2.g01 (geometry) ---

Geom Title=USGS 3m DEM
Program Version=4.10

River Reach=SpringCrk2      ,Main
Reach XY= 30
      1868660.82      659362.514     1869304.652      660044.947
     1867899.577      660711.789     1869073.507      663014.799
     1873087.591      662644.797     1871424.179      666046.895
     1872527.666       668145.39     1870932.197      667594.115
     1869890.008      668687.341     1870726.544       669873.38
     1869601.008      671867.134     1870474.775      672679.846
     1871101.458       671369.05     1873114.441      672977.122
     1872506.489      674496.768     1873519.039      674319.671
     1872327.517       676052.91     1873155.942       676389.89
     1872992.605      677869.617     1873946.011      679477.927
     1873487.475      679950.307      1871882.72      679385.765
     1873171.212      683022.659     1871587.207      684057.695
     1869301.583        682978.2     1870291.478      685566.888
     1867899.877      686379.565      1867555.71       691124.45
     1869386.358      689940.068     1869657.227      691117.628

Type RM Length L Ch R = 1 ,66291.3 ,359.7,362.6,365.6
XS GIS Cut Line= 4
     1868371.678      659673.079     1868672.544      659427.254
     1868798.226      659320.478     1870084.002      658335.095
#Sta/Elev= 30
       0  783.29   106.8  803.69   116.6  804.78   126.3   803.6   174.8   775.7
     272   733.6   301.1  723.18     340  718.45   378.8  706.38   407.9  704.92
   427.3  706.21   456.4  712.85   504.9   711.3   622.2  715.75   838.2  714.96
  1005.1  718.85  1181.8  715.82    1221  718.78  1270.1  725.22    1329   728.2
  1397.8  735.56  1446.9  738.89    1545  751.26  1574.5  751.46  1692.3   745.8
  1790.5  747.97  1967.2  761.18  2026.1  768.56  2134.1  794.81  2173.4  809.94
#Mann= 3 , 0 , 0
       0     .06       0   378.8    .045       0   427.3     .05       0
Bank Sta=378.8,427.3
XS Rating Curve= 0 ,0
Exp/Cntr=0.3,0.1

Type RM Length L Ch R = 1 ,65928.7 ,451.9,466.8,480.3
XS GIS Cut Line= 4
     1868378.106       659741.95     1868896.936      659693.602
     1869074.887      659576.415     1870240.252      658884.314
#Sta/Elev= 30
       0  772.21     177  786.74     236  790.74   255.6  790.46   285.1  782.66
   353.9  753.82   403.1   735.2   422.8  729.25   442.4  725.91   471.9  724.18
   521.1  717.75   588.9  706.18   598.6  705.08   617.9  706.73     647  712.33
   705.1  714.83  1136.8  714.68    1294  711.67  1352.9     718  1480.6  719.38
  1578.8  733.56  1667.2  748.71  1706.5  758.19  1755.6  774.39  1775.2  779.17
  1804.7  783.54  1834.2  785.48  1932.4  799.37  2001.1  815.15  2089.5  829.12
#Mann= 3 , 0 , 0
       0     .06       0   588.9    .045       0   617.9     .05       0
Bank Sta=588.9,617.9
XS Rating Curve= 0 ,0
Exp/Cntr=0.3,0.1

Type RM Length L Ch R = 1 ,65461.9 ,342.2,357.8,374.9
XS GIS Cut Line= 4
     1868427.524       659802.02     1869261.085      659931.189
     1869393.898      659933.793     1870094.419      659959.835
#Sta/Elev= 30
       0  766.61    88.3  770.99   186.4  771.19   304.1  774.68   402.1  753.02
   421.8  746.28   441.4  737.29   470.8  733.64   490.4  723.54   500.2  720.16
   725.8   719.6   804.3  717.85   833.7  715.55     872  706.89     891  704.71
   947.9  705.08   957.4  706.46   995.8  722.27  1044.5  754.88    1064   765.4
  1112.6  784.39  1161.3   806.6  1297.6  853.94  1346.3   867.1  1404.7  890.56
  1472.9  911.71    1541  926.04  1589.7  931.09  1609.2  929.45  1677.4  917.81
#Mann= 3 , 0 , 0
       0     .05       0     872    .045       0   957.4      .1       0
#XS Ineff= 2 , 0
          656.19  734.31
Permanent Ineff=
       F       F
#Block Obstruct= 1 ,-1
  541.81  653.18  765.56
Bank Sta=872,957.4
XS Rating Curve= 0 ,0
Exp/Cntr=0.3,0.1

Type RM Length L Ch R = 1 ,65104.1 ,374.4,386,397.2
XS GIS Cut Line= 4
     1868401.042      659877.026     1869060.565      660139.956
     1869182.092      660257.144     1869407.787      660521.901
#Sta/Elev= 30
       0  758.11    29.2  757.05    58.4  749.13    77.8  745.95   116.7  744.24
   126.4  744.94   145.9  748.25   165.3  749.52     214  747.07   291.8  738.18
   330.7  729.71   369.6  727.23     428     720   728.8  719.78   766.3  717.85
   775.7  715.77   794.4  706.54   803.8   704.7   822.6  706.06   831.9  708.74
   850.7  713.26   898.2  722.45   907.8  725.27   917.5  729.52  1004.5  779.68
  1062.4  809.35  1101.1  827.98  1197.7  858.02  1207.4  860.38  1226.7  863.31
#Mann= 3 , 0 , 0
       0     .05       0   775.7    .045       0   831.9      .1       0
#XS Ineff= 2 , 0
          738.39  721.47
Permanent Ineff=
       F       F
Bank Sta=775.7,831.9
XS Rating Curve= 0 ,0
Exp/Cntr=0.3,0.1

Type RM Length L Ch R = 1 ,64718.1 ,381.2,379.8,370.9
XS GIS Cut Line= 4
      1868330.15        659934.2     1868762.387      660300.546
      1868797.11      660413.394     1868900.118      660779.711
#Sta/Elev= 30
       0  747.62    48.8   744.9   166.1  741.65   195.4  734.48   214.9  730.99
   244.2  723.56   263.8  721.79   293.1  716.32   547.1  718.06   596.1  716.66
     606  715.04   615.8  711.92   625.6  707.88   635.5  705.27   645.3   704.7
     665   706.2   674.8  709.32   684.7   712.3   723.7   719.8   733.5  722.91
   743.2  727.98   762.7   740.8   821.3  781.08   840.8  795.89   850.5  801.82
   860.3  805.01   899.3   806.8   957.9  805.98   996.9  807.19  1065.2  803.63
#Mann= 3 , 0 , 0
       0     .05       0   615.8    .045       0   674.8      .1       0
Bank Sta=615.8,674.8
XS Rating Curve= 0 ,0
Exp/Cntr=0.3,0.1

Type RM Length L Ch R = 1 ,64338.3 ,405.6,400,392.5
XS GIS Cut Line= 3
     1868238.238      659980.356     1868409.188      660429.505
     1868718.559      660847.692
#Sta/Elev= 30
       0  733.74    19.6  740.08    39.2  743.48   156.9  742.24   176.5  738.24
   186.4  733.63     206  721.94   215.8  718.89     255  715.86   431.5  712.92
   451.2  708.96   470.8   704.7   490.4  705.02     510   710.1   549.3  720.85
   568.9   730.4   598.4  747.78   627.8  759.54   667.1  771.98   706.3  782.59
   784.8   799.5   804.5  800.26   833.9  799.12   922.2  793.01   932.1  791.66
   941.9  788.38   961.5   777.6   971.3  775.34   981.1  777.62  1000.8  786.55
#Mann= 3 , 0 , 0
       0     .05       0   451.2    .045       0     510      .1       0
Bank Sta=451.2,510
XS Rating Curve= 0 ,0
Exp/Cntr=0.3,0.1

Type RM Length L Ch R = 1 ,63938.3 ,94.2,87.6,90.2
XS GIS Cut Line= 3
     1867785.663      660147.018     1868018.163      660477.368
     1868640.373      660885.236
#Sta/Elev= 30
       0  806.32    28.8  811.06    57.7  813.45    96.2  811.75   134.6  807.31
   153.9  800.24   182.8  783.15     202  770.96   250.1  736.28   269.3  725.95
   288.6  718.51   365.5  707.04   394.4   704.7   413.8  704.98   433.3   708.5
   452.9  711.69   492.1  712.28   511.6  714.04   531.2  718.15   570.4  729.18
   629.1  739.18   678.1  743.84   746.6  746.43   873.8  761.64  1020.7  787.21
  1089.2  789.57    1099  788.11  1108.8  784.23  1138.2  764.88  1147.9  760.46
#Mann= 3 , 0 , 0
       0     .08       0   365.5    .045       0   433.3     .07       0
Bank Sta=365.5,433.3
XS Rating Curve= 0 ,0
Exp/Cntr=0.3,0.1

Type RM Length L Ch R = 1 ,63850.6 ,67.2,64.5,62.1
XS GIS Cut Line= 4
     1867667.769      660214.175     1867886.953      660481.102
     1867978.099      660552.717     1868590.078      660891.258
#Sta/Elev= 30
       0  797.41    28.8  803.81    76.8  808.88   105.5  809.47   134.3  805.16
   153.5  797.07   191.9  774.24   268.6  733.06   297.4  722.42   316.6  717.11
   345.4  714.72   374.4  709.13   393.7  705.55     413  704.74   422.7  705.12
     442  709.38   461.3  711.88   509.9  711.28   529.3  713.84   548.7  717.61
   587.6  728.32   645.9  739.14   733.3  744.96     811  744.87   859.6  748.39
   966.4  763.66  1102.4  786.83  1121.8  788.37  1141.2   787.5  1160.7  780.59
#Mann= 3 , 0 , 0
       0     .08       0   374.4    .045       0     442     .07       0
Bank Sta=374.4,442
XS Rating Curve= 0 ,0
Exp/Cntr=0.3,0.1

Type RM Length L Ch R = 1 ,63786.1 ,51.1,48.7,45.8
XS GIS Cut Line= 4
     1867453.794      660268.862      1867826.19      660528.845
     1867992.856       660631.71     1868539.731      660897.335
#Sta/Elev= 30
       0  774.21      29  763.83    77.3  742.41    96.6  735.63     116  731.12
   135.3  730.91   173.9  735.24   241.6  747.82   260.9  748.99   280.2  746.86
   328.6  737.41   367.2  723.93   386.5  720.27   512.9  708.01   542.3  704.71
   571.7   708.9   601.1  712.28   640.2  711.66   669.6  713.89   689.2  718.74
   708.9  727.62   728.5  734.13   748.1  737.95   846.1  745.12   944.2  742.51
    1003  745.22  1130.5  763.82  1218.8   780.2  1238.4   782.7    1258  782.46
#Mann= 3 , 0 , 0
       0     .08       0   512.9    .045       0   571.7     .08       0
Bank Sta=512.9,571.7
XS Rating Curve= 0 ,0
Exp/Cntr=0.3,0.1

Type RM Length L Ch R = 1 ,63737.5 ,184.7,176,167.9
XS GIS Cut Line= 4
     1867348.759      660387.786     1867852.231       660606.97
     1867971.589      660661.224     1868529.315      660916.432
#Sta/Elev= 30
       0  805.45    68.6  783.83    98.1  770.71   176.5  739.77   205.9  725.91
   225.5  719.69   313.8   721.8     353  721.45     402   716.3   480.5  715.16
   529.5  712.51   549.1  710.34   567.8  706.04   586.6   704.7   614.7  704.92
   633.4  706.86   652.1  710.15     690     712   709.4  714.85   728.9  718.98
   767.8  731.37     797   737.6   894.4  743.96   991.8  741.55  1050.2  744.19
  1079.4  747.45  1186.5  763.58  1264.4  778.15  1283.8  779.39  1293.6  777.56
#Mann= 3 , 0 , 0
       0     .08       0   567.8    .045       0   633.4     .08       0
Bank Sta=567.8,633.4
XS Rating Curve= 0 ,0
Exp/Cntr=0.3,0.1

Type RM Length L Ch R = 1 ,63561.4 ,452.3,442.5,432.1
XS GIS Cut Line= 4
      1867182.96      660789.696     1867832.266       660796.64
     1867988.516      660807.057     1868516.294      660938.133
#Sta/Elev= 30
       0  822.96    78.7  814.56   196.8     807     246  800.41   285.3  793.04
   314.8  784.73   324.7  780.59   344.4  768.32   383.7  736.79   393.5  730.03
   403.4  725.46   413.2   723.3   452.6  718.47   472.2  717.13   708.1  711.08
     722   709.3   737.4  705.71   747.2   704.7   776.6   704.9   796.2   708.7
   815.6  711.88   893.3  716.17   961.3   729.1  1019.6  736.47  1097.3   739.5
  1145.8  743.26  1262.4  761.04  1330.3  774.67    1340  774.12  1349.8   771.2
#Mann= 3 , 0 , 0
       0     .08       0     722    .045       0   796.2     .08       0
Bank Sta=722,796.2
XS Rating Curve= 0 ,0
Exp/Cntr=0.3,0.1

Type RM Length L Ch R = 1 ,63118.9 ,387.9,381.2,374.4
XS GIS Cut Line= 4
     1867511.953      661426.415     1867988.516       661236.31
      1868147.37      661168.602     1868571.849       661035.79
#Sta/Elev= 30
       0  856.87      29   845.2    48.4  840.05    87.1  845.45   125.8  846.56
   164.6  843.74   193.6  837.64   222.7  828.05   290.4  800.12   309.8  789.95
   358.2  760.07   387.2  748.38   464.7  723.45   493.7  717.56   541.9  712.94
     561  707.59   570.6  705.22   589.8   704.7   618.6  705.01   628.2  706.73
   647.4  709.52   879.1  714.88   908.2   717.8   937.2  724.66   946.8  725.48
   975.8  723.86   995.2  724.58  1062.8  732.76  1101.5  748.42  1130.5  753.44
#Mann= 3 , 0 , 0
       0      .1       0     561    .045       0   628.2      .1       0
Bank Sta=561,628.2
XS Rating Curve= 0 ,0
Exp/Cntr=0.3,0.1

Type RM Length L Ch R = 1 ,62737.7 ,399.9,398.2,396.4
XS GIS Cut Line= 5
     1867017.548      662134.547     1867660.482      661940.939
     1868261.719      661530.153     1868389.558      661426.849
      1868694.93      661153.055
#Sta/Elev= 30
       0  841.97    48.7  856.07   155.7  893.04   282.2  913.56   311.4  915.64
   389.2   904.1   476.8  878.49   515.8  872.16   564.4  871.48   622.8  874.42
   671.4  871.29   779.7  872.98   956.8  868.24    1006  859.47  1183.1  798.37
  1242.2  774.46  1291.4   762.2  1340.6   741.7  1370.1  734.63  1409.3  718.65
  1457.6  705.81  1475.8   704.7  1515.6  706.57    1535   709.8  1710.5   715.7
    1730  721.74  1827.6  766.73  1866.7  779.37  1925.3  789.32  1974.1  793.42
#Mann= 3 , 0 , 0
       0      .1       0  1457.6    .045       0  1515.6      .1       0
Bank Sta=1457.6,1515.6
XS Rating Curve= 0 ,0
Exp/Cntr=0.3,0.1

Type RM Length L Ch R = 1 ,62339.6 ,414,423.8,433.7
XS GIS Cut Line= 5
     1867429.875       663065.97     1868047.541      662501.697
     1868582.849      661758.207     1868704.662      661642.994
     1868977.109       661349.85
#Sta/Elev= 30
       0  829.22    88.6  791.31   137.8  761.84   157.5   764.4     187  781.64
   216.5  794.31   295.3  817.02   324.8  813.62   383.9  795.37   482.3  833.03
     502  835.15   708.7  818.95   807.1  803.07   865.8  789.91   953.6  761.84
   992.6  753.71  1031.5  739.53  1148.5  719.49  1216.7  715.91  1577.3   715.1
  1836.6  706.88  1862.6   704.7  1892.5   704.7  1911.1  707.55    1979  712.14
    2018  739.97  2066.8  769.74  2105.9  792.14  2125.4  799.79  2320.6  822.61
#Mann= 3 , 0 , 0
       0     .06       0  1836.6    .045       0  1911.1      .1       0
#XS Ineff= 2 , 0
         1722.41  721.62
Permanent Ineff=
       F       F
Bank Sta=1836.6,1911.1
XS Rating Curve= 0 ,0
Exp/Cntr=0.3,0.1

Type RM Length L Ch R = 1 ,61915.7 ,403.6,403.8,404
XS GIS Cut Line= 4
     1868183.828      662473.724     1868662.995      662111.744
     1868910.391      662031.015      1869268.05      661994.369
#Sta/Elev= 30
       0  786.53    48.4  769.32    96.9  759.19   135.6     746   145.3  743.42
   251.8  727.02     310  719.45   348.7  717.37   600.5  716.06   706.6  712.68
   716.2  711.93   725.8  709.51   735.5  706.33   745.1  704.93   754.7   704.7
   783.6  704.85   793.3  706.24   802.9  710.39   851.1  741.66   870.5  753.42
   880.2  758.04   889.9  761.46   899.6   763.7   948.2  770.25  1006.5  784.12
  1035.7  789.18  1055.1  791.01  1113.4  794.19  1152.3  795.18  1220.3  798.92
#Mann= 3 , 0 , 0
       0     .06       0   725.8    .045       0   802.9      .1       0
#XS Ineff= 2 , 0
          600.45  718.07
Permanent Ineff=
       F       F
Bank Sta=725.8,802.9
XS Rating Curve= 0 ,0
Exp/Cntr=0.3,0.1

Type RM Length L Ch R = 1 ,61511.9 ,370.4,368.8,367.2
XS GIS Cut Line= 4
      1868366.12      662623.029     1868806.658       662477.63
     1868917.102      662441.996     1869214.644      662345.251
#Sta/Elev= 30
       0  793.39    19.3  788.54    38.7  781.73    48.3  777.39      87  758.05
   106.3  749.74     116  746.13   154.6  735.88   212.6  721.88   222.3  720.59
   280.3  718.77   454.2  711.44   463.9  710.39   473.6  707.97   483.2  705.32
   492.9   704.7   531.6  704.94   541.3  706.28     551  708.36   589.7  714.05
   599.5  716.66   628.8  729.72   648.4  735.82   677.7  742.89   716.8  751.42
     756  758.82   775.5   761.9     844  770.26   863.5  771.15   892.8  769.61
#Mann= 3 , 0 , 0
       0     .06       0   473.6    .045       0     551      .1       0
Bank Sta=473.6,551
XS Rating Curve= 0 ,0
Exp/Cntr=0.3,0.1

Type RM Length L Ch R = 1 ,61143.1 ,252.3,236.9,221.2
XS GIS Cut Line= 4
      1868527.55      662933.669     1868906.485      662835.703
     1869030.183       662785.79     1869281.919      662462.439
#Sta/Elev= 30
       0  837.93     9.8  830.56    19.6  824.57    29.4  820.04    58.7  808.47
    78.3  800.16   117.4   780.1     137  769.49   156.6  757.96   195.7  732.19
   215.3  722.08     225  718.31   234.8   716.9   244.6  716.26   381.6  708.81
   391.4   707.8   410.4  704.77     420   704.7   458.1  704.92   477.1  707.46
   486.7  708.36   534.5  710.44   671.1  717.77   680.9  719.04     759  732.24
   827.2  742.46     876  748.11   895.5  749.81   915.1  751.02   934.6  751.04
#Mann= 3 , 0 , 0
       0     .05       0   391.4    .045       0   477.1     .06       0
Bank Sta=391.4,477.1
XS Rating Curve= 0 ,0
Exp/Cntr=0.3,0.1

Type RM Length L Ch R = 1 ,60906.2 ,230,215.9,202
XS GIS Cut Line= 4
      1868826.19      663510.616     1869004.141      663143.862
     1869130.009      662915.998     1869338.342        662479.8
#Sta/Elev= 30
       0   801.1    19.4  792.08    48.5  775.03    67.9  767.04    77.6  765.16
   106.8  765.76   116.5  768.82   145.6  783.03   194.1  802.07   242.6  816.62
   252.4  818.81   262.1  819.22   281.5  811.16   291.2  805.24   320.3  783.43
   339.7  770.36   407.6  732.22   417.3  728.92   494.4  712.95   513.7  706.61
     533   704.7   571.6  704.72   590.8  706.25   648.7  708.88   822.6  711.65
     871  715.22   996.7  730.73  1112.7  741.85    1132  742.31  1151.4  739.81
#Mann= 3 , 0 , 0
       0     .07       0   513.7    .045       0   590.8     .05       0
Bank Sta=513.7,590.8
XS Rating Curve= 0 ,0
Exp/Cntr=0.3,0.1

Type RM Length L Ch R = 1 ,60690.3 ,352.1,352,350.9
XS GIS Cut Line= 4
      1869363.57      663438.075      1869291.12      663060.327
     1869273.759      662914.493     1869416.015      662504.967
#Sta/Elev= 30
       0  878.96    28.8  857.38    38.5  852.28    48.1  849.32    67.3  844.99
    76.9  841.05   115.4  820.23   144.2  809.99   153.8   805.1   163.5  797.84
   182.7  781.44   192.3  774.78   259.6  738.72   269.2  734.81   278.9  732.39
   365.4  717.34   394.4   711.3   404.2  708.19     414  705.43   423.8   704.7
     463  704.74   482.5  707.52   560.4  709.51   695.3  714.49   714.5  717.15
   753.1  724.64   772.4  726.69   878.3  729.38   936.1  725.45     965  722.57
#Mann= 3 , 0 , 0
       0     .07       0   404.2    .045       0   482.5     .05       0
Bank Sta=404.2,482.5
XS Rating Curve= 0 ,0
Exp/Cntr=0.3,0.1

Type RM Length L Ch R = 1 ,60338.3 ,398,400,401.2
XS GIS Cut Line= 3
     1869684.833      663397.956     1869628.431      662946.548
      1869553.42        662497.3
#Sta/Elev= 30
       0  851.47    38.7  846.12    48.4  844.08    58.1  840.21   116.2  809.26
   125.8   802.7   154.9   780.4   164.5  774.65   193.6  762.11   222.6  748.59
   232.3  745.37   290.4  730.79   348.4  713.87   367.8   711.4   406.5  708.46
   416.2  706.79   425.9  704.77   435.6   704.7   474.3  704.71     484  705.15
   493.7  706.76   561.5  706.31     610  710.32   668.1  712.89   677.8  714.44
   726.3  727.21   755.3  735.72     765  737.64   794.1  740.71   910.4  747.36
#Mann= 3 , 0 , 0
       0     .05       0   416.2    .045       0   493.7     .05       0
Bank Sta=416.2,493.7
XS Rating Curve= 0 ,0
Exp/Cntr=0.3,0.1

Type RM Length L Ch R = 1 ,59938.3 ,415.1,400,386.8
XS GIS Cut Line= 3
     1870032.969       663312.53     1870016.563      662857.927
     1869966.655       662403.11
#Sta/Elev= 30
       0  826.69     9.7  823.45    38.7  807.94    96.8  773.55   212.9   723.3
   232.3  716.98   261.3  712.48   319.4  707.95   358.1  707.11   396.8  708.56
   406.5  708.45   416.2  707.24   425.9   705.3   435.5   704.7   474.4   704.7
   484.1   705.1   493.8  706.88   503.6  708.39   542.5  707.51   600.9  708.39
   620.4  710.59   630.1  712.72   639.9  716.13   649.6  721.68   669.1  734.95
   678.8  739.49   698.3  745.12   727.5  751.04   873.5  775.16   912.4  780.59
#Mann= 3 , 0 , 0
       0     .05       0   416.2    .045       0   493.8    .055       0
Bank Sta=416.2,493.8
XS Rating Curve= 0 ,0
Exp/Cntr=0.3,0.1

Type RM Length L Ch R = 1 ,59538.3 ,390.6,400,409.2
XS GIS Cut Line= 3
      1870658.11      663064.837     1870358.638        662714.4
     1870069.747      662360.968
#Sta/Elev= 30
       0  762.19     9.8  757.91    29.4  750.19   107.9  720.39   117.7  717.29
   127.5  715.14   137.3  713.79   156.9  712.01   284.4  707.09   323.7  707.14
   402.1  708.29   411.9  707.67   421.7  705.49   431.5  704.71   441.4   704.7
   480.4  704.77   499.8  706.58   558.1  709.88   567.8   710.8   577.5  712.97
   587.2  718.29   606.6  730.77   626.1   742.5   635.8  746.59   645.5  749.35
   684.4  757.32   742.6  767.87     830  784.48   888.3  798.23   917.4  802.93
#Mann= 3 , 0 , 0
       0     .05       0   411.9    .045       0   499.8     .08       0
Bank Sta=411.9,499.8
XS Rating Curve= 0 ,0
Exp/Cntr=0.3,0.1

Type RM Length L Ch R = 1 ,59138.3 ,558.8,562.1,565.1
XS GIS Cut Line= 3
     1870850.624       662997.79     1870718.768      662563.117
     1870593.845       662122.53
#Sta/Elev= 30
       0  764.84    19.3  757.17      87  728.68   106.3  721.07     116  717.56
   125.6   714.6     145  710.87   154.6  709.63   164.3  709.07   270.6  706.11
   405.9  706.69   415.6  706.45   434.9   704.7     503  704.76   512.7  709.17
   522.4  715.29   532.2  720.42   551.7  728.27   561.4  731.54   571.2  733.52
   610.1  737.13   649.1  741.61   697.8  745.42   727.1  748.33   746.5  750.88
     766     754   834.2  769.84   853.7  775.23   873.2  781.98   912.2  796.77
#Mann= 3 , 0 , 0
       0     .05       0   415.6    .045       0   512.7      .1       0
Bank Sta=415.6,512.7
XS Rating Curve= 0 ,0
Exp/Cntr=0.3,0.1

Type RM Length L Ch R = 1 ,58576.2 ,188.7,189.6,189.3
XS GIS Cut Line= 4
     1871334.848      663019.202     1871277.557      662576.494
     1871260.476       662460.45     1871167.748      661840.817
#Sta/Elev= 30
       0  811.42    58.2  809.04   126.2   803.4   135.9  801.57   155.3  793.81
   232.9  757.24   349.4  715.39   359.1  712.87   378.5  709.38   436.7  706.26
   446.4  704.89   456.2   704.7   514.8  704.74   524.6   706.4   534.4  707.01
   612.6  706.89   651.8   707.5   749.7   711.8   769.3  713.66   779.1  717.15
   798.6     728   808.4  732.79     828  739.31   847.6  744.45   955.3     765
  1004.2  775.12  1072.8  787.77  1141.3  802.61  1170.6     808  1190.2   810.6
#Mann= 3 , 0 , 0
       0     .06       0   436.7    .045       0   524.6     .05       0
Bank Sta=436.7,524.6
XS Rating Curve= 0 ,0
Exp/Cntr=0.3,0.1

Type RM Length L Ch R = 1 ,58386.6 ,47.8,47.8,47.8
XS GIS Cut Line= 5
     1871526.037      662994.921     1871468.203      662596.785
      1871453.57      662487.454     1871429.466      662280.921
     1871515.404      661804.359
#Sta/Elev= 30
       0  804.48    29.4  805.24    88.3  804.77   137.4  801.34   166.8  798.42
   176.6  795.73   235.5  768.51   255.1  760.09   294.4   745.9   304.2  741.91
     314  736.29   343.4   715.4   353.2  711.74   392.5  709.67   402.3  708.73
   420.7  705.27   429.9  704.72   475.8   704.7   494.2  704.71   588.2  705.23
   759.3  708.92   846.5  712.92     982  713.67    1108  718.69  1127.3  720.45
    1137  722.58  1146.7  726.27  1185.4  746.04  1195.1  750.12  1204.8  753.45
#Mann= 3 , 0 , 0
       0     .06       0   420.7    .045       0   494.2     .06       0
#XS Ineff= 2 , 0
                          674.25          717.35
Permanent Ineff=
       F       F
Bank Sta=420.7,494.2
XS Rating Curve= 0 ,0
Exp/Cntr=0.3,0.1

Type RM Length L Ch R = 1 ,58338.8 ,173.5,175.6,177.6
XS GIS Cut Line= 5
     1871572.912      662984.504     1871515.078      662586.368
     1871500.445      662477.038     1871476.341      662270.505
     1871554.466      661814.775
#Sta/Elev= 30
       0  795.51    29.4  799.08    78.5  800.74   107.9  799.39   137.4  795.44
     157  793.79   166.8  791.94   196.2  782.96   235.5   767.1   294.4   746.1
   304.2  741.78     314  735.44   333.6  720.12   343.4  713.48   353.2  709.76
   372.9  707.49   402.3  707.85   420.7  703.01   466.7   702.8   475.8  702.81
   494.2  706.71   531.5  706.39   588.2  708.17   740.2  710.48   966.5  716.12
  1064.9  720.53  1074.7     722  1084.6  724.69  1143.6  751.43  1182.9  762.67
#Mann= 3 , 0 , 0
       0     .06       0   402.3    .045       0   494.2     .05       0
#XS Ineff= 2 , 0
                          634.11          716.76
Permanent Ineff=
       F       F
Bank Sta=402.3,494.2
XS Rating Curve= 0 ,0
Exp/Cntr=0.3,0.1

Type RM Length L Ch R = 1 ,58163.2 ,224.8,228.6,232.5
XS GIS Cut Line= 4
     1871686.411       662929.72     1871682.071      662593.349
      1871673.39      662411.057      1871731.55      661839.877
#Sta/Elev= 30
       0   762.5    38.4  765.47    96.1   758.6   201.8  757.27   221.1  755.38
   249.9  748.28   269.1  741.58   278.7  735.71   307.6  715.03   317.2  710.37
   326.8  708.08   336.4  707.19   384.4  706.39     394  704.81   403.6  701.57
   413.2  699.96   451.7  701.05   470.9  704.82   490.1  706.69   625.9  709.49
   771.9  714.01   859.5  713.35     879  713.72   898.4  715.62   927.6  720.37
   937.3  723.32   976.3  740.93  1005.4  750.68  1073.6  778.36    1093  784.27
#Mann= 3 , 0 , 0
       0     .05       0     394    .045       0   470.9     .05       0
Bank Sta=394,470.9
XS Rating Curve= 0 ,0
Exp/Cntr=0.3,0.1

Type RM Length L Ch R = 1 ,57934.6 ,392.5,387.5,382.5
XS GIS Cut Line= 4
     1871832.535      662941.816     1871895.612      662558.627
      1871921.26       662363.67     1871991.966      661811.231
#Sta/Elev= 30
       0  745.79    29.1  740.51    58.2  738.77   106.8  741.84   174.8   740.2
   252.4  743.62   262.1  741.85   271.8  738.13     301  720.51   310.7  715.41
   320.4  711.58   330.1  709.08   349.5  706.95   398.2  705.45     408  704.38
   417.8  701.62   427.7   699.1   437.5   698.4     467  698.41   476.8  699.52
   486.7  702.32   496.5  704.72   506.3  705.52   809.7  712.84   985.6  721.14
   995.4  723.82  1073.5  768.02  1083.3  772.36  1102.8  777.25  1141.9  784.56
#Mann= 3 , 0 , 0
       0     .05       0   417.8    .045       0   486.7     .05       0
Bank Sta=417.8,486.7
XS Rating Curve= 0 ,0
Exp/Cntr=0.3,0.1

Type RM Length L Ch R = 1 ,57547.1 ,404.8,405.1,405.4
XS GIS Cut Line= 4
     1872281.105      662943.651     1872283.633       662516.96
     1872268.008      662342.481     1872202.904      661795.606
#Sta/Elev= 30
       0  754.48    77.6  751.76   242.4  751.73   290.9  750.39   339.4  748.29
   349.1  745.53   358.8   740.1   387.9  720.91   397.6  716.68     417  711.59
   436.4  707.75   446.2  703.93   455.9  699.96   465.6  698.54   475.4   698.4
   504.6  698.42   514.3  699.63     524  702.19   533.8  703.89   543.5  704.35
   690.4   707.1   847.7  712.24   975.6   719.4   985.4  721.09  1014.9  732.39
  1034.6  736.76  1064.1  749.49  1083.8  756.19  1093.6  758.12  1152.6  765.61
#Mann= 3 , 0 , 0
       0    .065       0   446.2    .045       0     524     .05       0
Bank Sta=446.2,524
XS Rating Curve= 0 ,0
Exp/Cntr=0.3,0.1

Type RM Length L Ch R = 1 ,57141.9 ,253.1,264.4,275.5
XS GIS Cut Line= 4
      1872369.66      662923.313     1872650.821      662404.981
     1872622.175      662165.397     1872583.112       661735.71
#Sta/Elev= 30
       0  751.23    39.3  753.21    98.3   753.7   275.2  750.98   294.8  749.83
   353.8  744.13   373.5  741.04     403  734.48   422.6   728.9   461.9  713.89
   471.7  711.17   491.4  709.73   657.2   705.5   666.9   704.9   676.5  702.96
   686.2  700.24   695.8  698.69   705.5   698.4   744.1   698.6   763.4  702.87
     831  701.19   870.2  705.02   889.8  705.97   899.6   707.1   909.4  709.77
   948.6   726.9  1027.1  757.27    1135  795.06  1213.4  825.41  1262.4  839.81
#Mann= 3 , 0 , 0
       0     .05       0   676.5    .045       0   763.4    .065       0
Bank Sta=676.5,763.4
XS Rating Curve= 0 ,0
Exp/Cntr=0.3,0.1

Type RM Length L Ch R = 1 ,56877.6 ,338.6,356.4,374.2
XS GIS Cut Line= 4
     1872443.403      662948.637     1872747.175      662519.564
      1872919.05      662126.335     1873096.133       661766.96
#Sta/Elev= 30
       0  751.84   223.9  750.75   253.1  749.54   292.1  743.18   399.2  729.44
   457.6   724.2   467.3  721.63   506.2  707.81     516  706.76   652.5  707.35
   798.8  705.15   808.6  704.67   818.3  702.28   828.1  699.43   847.6   698.4
   876.8   698.6   886.6  701.21   896.4  709.02   915.9  732.04   925.6  740.32
     994  782.48  1072.1  824.99  1101.4   838.4  1140.5  850.85  1218.7  873.96
  1257.8  880.17  1267.6   883.3  1277.3  889.04  1316.4  915.45  1355.5  935.57
#Mann= 3 , 0 , 0
       0     .05       0   818.3    .045       0   886.6      .1       0
Bank Sta=818.3,886.6
XS Rating Curve= 0 ,0
Exp/Cntr=0.3,0.1

Type RM Length L Ch R = 1 ,56521.2 ,585.7,594.8,603.8
XS GIS Cut Line= 3
     1872484.911      663032.652     1872934.675      662576.856
       1873512.8      662347.689
#Sta/Elev= 30
       0   749.5    77.6  750.52   155.2  747.73   164.9  746.92   184.3  744.04
   252.3  730.44   281.4  725.58     359  717.38   388.1  715.08   514.2  708.43
   582.1  705.44   708.4  704.58   718.1  704.11   727.8   702.2   737.5  699.49
   747.2   698.5     757   698.4   786.1   698.5   795.8  699.48   805.5  702.48
   883.3  742.38   902.7  751.92   922.1  760.79     961  777.56   990.2  788.79
  1116.5     840  1194.2  867.78  1213.6  873.53  1242.8  880.76  1262.2  887.09
#Mann= 3 , 0 , 0
       0     .05       0   727.8    .045       0   805.5      .1       0
Bank Sta=727.8,805.5
XS Rating Curve= 0 ,0
Exp/Cntr=0.3,0.1

Type RM Length L Ch R = 1 ,55926.3 ,381,388,396.9
XS GIS Cut Line= 4
     1872475.147      663124.777     1872853.946      663087.272
     1873025.759       663090.27     1873497.175      663128.939
#Sta/Elev= 30
       0  743.62     9.8  744.65      39  745.03   126.9  743.69   136.6  741.76
   156.2  735.14   165.9   732.6   185.4  728.08   224.5  717.51   234.2  715.77
   253.8  714.36   390.2  707.38   409.3  705.28   418.8  702.42   428.4  699.14
   437.9  697.61   447.5   697.6   485.7  698.22   495.2  698.72   504.8  699.96
   600.8  717.48   639.4  726.37   697.3  741.07   784.2  768.01   793.8  771.59
   803.5  776.37   813.1  782.05   890.4  828.84   977.2  871.61  1025.5  899.82
#Mann= 3 , 0 , 0
       0     .05       0   418.8    .045       0   504.8      .1       0
Bank Sta=418.8,504.8
XS Rating Curve= 0 ,0
Exp/Cntr=0.3,0.1

Type RM Length L Ch R = 1 ,55538.3 ,397,400,401.2
XS GIS Cut Line= 3
     1872458.713      663323.321     1872890.946      663471.121
     1873307.911      663652.436
#Sta/Elev= 30
       0  743.05    58.3  738.99    87.5  734.98   106.9  731.17   136.1  721.56
   145.8  718.95   155.5  717.27   194.4  713.67   233.3  711.11   252.7  710.39
   281.9  710.32   320.7  706.96   388.8  702.91   398.5  701.94   408.2  700.24
   417.9  698.45   427.6  697.57   437.4   697.5   485.8  698.35   495.5  699.84
   505.2  703.93   514.8  709.99   543.9  730.05   592.2  759.88   621.3  775.66
   708.3  820.94     718  825.16   843.8  863.33   863.1  867.56   911.5  874.76
#Mann= 3 , 0 , 0
       0     .05       0   408.2    .045       0   495.5      .1       0
Bank Sta=408.2,495.5
XS Rating Curve= 0 ,0
Exp/Cntr=0.3,0.1

Type RM Length L Ch R = 1 ,55138.3 ,393,397.6,402
XS GIS Cut Line= 3
     1872318.748      663631.602     1872725.712      663835.085
     1873132.676      664038.567
#Sta/Elev= 30
       0  771.54    38.7  763.98   106.5   749.6   116.2  746.78   125.8  743.45
   164.6  729.18   183.9  721.81   193.6   719.6     242  714.54   300.1  709.01
   396.9  704.42   406.6  703.31   416.3  700.24     426  697.54   435.6   697.1
   474.4  697.76     484   699.1   493.7  702.59   503.4  707.11   532.4  719.69
   590.5  743.68   648.6  768.18     668  775.78   687.3  781.95   764.8  804.99
   774.5  807.33   803.5  813.59   842.2  821.66   851.9  823.29     910  829.67
#Mann= 3 , 0 , 0
       0     .05       0   406.6    .045       0   493.7      .1       0
Bank Sta=406.6,493.7
XS Rating Curve= 0 ,0
Exp/Cntr=0.3,0.1

Type RM Length L Ch R = 1 ,54740.7 ,269.8,281.4,293
XS GIS Cut Line= 5
     1872166.956      663916.871     1872481.116      664140.658
     1872595.323      664229.943     1873132.157      664257.845
     1873456.784      664125.866
#Sta/Elev= 30
       0  783.44    28.9  778.52    57.9  771.27   192.9  728.39   212.1  723.33
   298.9  706.88   337.5  704.14   385.7  703.96     405  701.18   414.7  697.53
     434   696.3   472.7  696.87     492  700.19   501.7  703.64     521  706.41
   569.8  708.85   608.9  712.56   628.4  719.71   677.3  744.91   706.6  756.16
   814.1  787.51     863  805.84   882.5  809.94   911.9  813.03   980.3  815.36
  1029.2  813.82  1068.2  809.31  1126.6  808.56  1301.9  792.99  1418.7  789.87
#Mann= 3 , 0 , 0
       0     .05       0     405    .045       0     492     .07       0
Bank Sta=405,492
XS Rating Curve= 0 ,0
Exp/Cntr=0.3,0.1

Type RM Length L Ch R = 1 ,54459.4 ,73.9,79.3,84.8
XS GIS Cut Line= 5
     1872157.765      663945.345     1872300.994      664286.057
     1872374.779      664461.838     1872876.081      664963.141
     1873710.257      665077.255
#Sta/Elev= 30
       0  781.36    29.2  776.55   136.2  750.05   194.5  733.24   223.7  721.21
   243.2  716.23   330.7  703.98   369.6  702.18   417.2  702.52   436.3  699.02
   445.8  696.58   464.9  696.12   531.6  696.92   560.2  699.57   764.2  703.52
   773.9  705.09   822.4  721.92   890.4  734.67   977.8  744.63  1026.4  755.89
    1075  763.16  1142.9  778.31  1210.9  799.56  1269.2  806.47  1357.3  810.37
  1533.5  811.95  1641.2   821.2  1827.2  831.52  1983.8  832.35  2111.1  827.58
#Mann= 3 , 0 , 0
       0     .05       0   436.3    .045       0   560.2     .07       0
Bank Sta=436.3,560.2
XS Rating Curve= 0 ,0
Exp/Cntr=0.3,0.1

Type RM Length L Ch R = 1 ,54380.1 ,77,77.4,79.1
XS GIS Cut Line= 5
     1872136.064      663954.026     1872268.384      664373.282
     1872296.654      664516.092     1872322.696      664713.575
     1872559.241       664954.46
#Sta/Elev= 30
       0  779.56    48.8  772.21     127  753.45   156.3  744.31   195.4  729.75
   214.9  721.23   224.7  718.14   234.5  716.19   244.2  715.16     254  715.04
   302.9   715.4   361.5  707.92   429.9  697.46   439.6  696.26     459  696.03
   517.3  696.44   536.7  697.77   556.1  700.25   585.2  705.31   613.7  707.21
   642.1  707.37   689.6  705.32     737  704.67   784.4  706.04   871.2  706.33
   919.5  717.31   977.3  734.82  1006.3  742.18  1083.4  767.92    1122  779.76
#Mann= 3 , 0 , 0
       0     .07       0   429.9    .045       0   536.7     .05       0
Bank Sta=429.9,536.7
XS Rating Curve= 0 ,0
Exp/Cntr=0.3,0.1

Type RM Length L Ch R = 1 ,54302.7 ,168.5,166.3,162.7
XS GIS Cut Line= 5
       1872075.3      663993.088      1872207.62      664412.344
      1872235.89      664555.154     1872261.932      664752.637
     1872498.477      664993.522
#Sta/Elev= 30
       0  769.25    39.1   763.2    97.7  748.69   107.5  745.38   136.8  730.22
   146.6  726.77   156.3  725.96   166.1  726.96   185.6  732.48   205.2  735.34
   302.9  729.68   312.6  728.66   371.2  717.29   400.6  709.64   420.1  705.95
   439.6  700.02     459   696.5   488.2     696   536.7  696.44   556.1   699.1
   575.5  703.04   594.7  704.79   708.5  704.72     756  703.38     823  706.94
   909.8  709.34   929.1  713.07   967.7  725.12  1054.5  756.46    1122  779.16
#Mann= 3 , 0 , 0
       0     .07       0   439.6    .045       0   556.1     .05       0
Bank Sta=439.6,556.1
XS Rating Curve= 0 ,0
Exp/Cntr=0.3,0.1

Type RM Length L Ch R = 1 ,54136.3 ,212.7,192.6,172.1
XS GIS Cut Line= 4
     1871832.244      664084.234     1872092.661      664544.304
     1872216.359      664780.849     1872483.286      665002.203
#Sta/Elev= 30
       0     792    58.7  782.11   156.6  770.62   205.6  762.35   254.5   756.5
   283.9  752.26   332.9  747.76     372   740.8   469.9  725.43   509.1  721.64
   518.9  719.27   528.7  715.41   547.7  706.03   557.3   702.2   566.8  699.14
   576.3  697.27   585.9  695.82   604.9   694.7   643.1  695.58   652.6  696.48
   662.1  698.13   671.7  699.58   681.2   700.2   757.5  701.37   949.7  711.06
   959.4  712.58   978.6  718.68  1055.7  747.57  1094.2  762.74  1142.4  778.57
#Mann= 3 , 0 , 0
       0     .08       0   576.3    .045       0   662.1     .06       0
Bank Sta=576.3,662.1
XS Rating Curve= 0 ,0
Exp/Cntr=0.3,0.1

Type RM Length L Ch R = 1 ,53943.7 ,407.4,399.6,391.6
XS GIS Cut Line= 4
     1871660.122      664633.214     1872042.748      664789.529
     1872153.028      664841.293     1872485.456      665021.734
#Sta/Elev= 30
       0  801.52    39.4   777.9    49.2  773.04    78.7  762.07    98.4  755.51
   108.2  753.49   127.9  751.01   137.8  748.52   157.5  742.15   206.7  728.86
   226.3  724.63   236.2  723.41   364.1  710.31   432.1  695.67   450.8     693
   469.6  692.43   478.9   692.6   488.3  693.86   497.7  697.49     507  699.74
   516.4  700.58   593.3  704.85   670.9  707.66     700  709.63   709.7  710.86
   719.4  712.98   729.1  716.38   777.6   736.6   855.2   766.4   913.4  784.44
#Mann= 3 , 0 , 0
       0     .08       0   432.1    .045       0   497.7     .08       0
Bank Sta=432.1,497.7
XS Rating Curve= 0 ,0
Exp/Cntr=0.3,0.1

Type RM Length L Ch R = 1 ,53544.1 ,392.6,407.6,422.6
XS GIS Cut Line= 4
     1871469.831      665073.818     1871938.353      665170.928
     1872133.894      665188.835     1872439.883      665227.897
#Sta/Elev= 30
       0  773.04    19.5   764.9    48.8  753.77    87.9  737.42    97.6  734.11
   107.4  732.12   136.7  728.61   185.5  721.55   214.8  717.82   234.4  714.12
   253.9  711.99   322.2  707.15   351.5  705.61   449.2   702.2   576.7  693.11
   606.1   692.4   625.8   692.6   635.6  693.79   655.2  698.58     665  700.42
   674.8  703.18   684.5  707.17   742.3  734.17   771.2  745.92   829.1  767.41
   867.6  779.57   925.5  799.95   935.1  802.65   944.8  804.39   983.3  809.03
#Mann= 3 , 0 , 0
       0     .08       0   576.7    .045       0   635.6     .08       0
Bank Sta=576.7,635.6
XS Rating Curve= 0 ,0
Exp/Cntr=0.3,0.1

Type RM Length L Ch R = 1 ,53136.5 ,406,401.3,396.2
XS GIS Cut Line= 4
     1871419.918      665158.453     1871801.897       665479.31
     1871899.519      665570.779     1872298.824      665883.279
#Sta/Elev= 30
       0  777.13    39.1  759.91    48.9  755.94    68.5  748.89    97.8  740.12
   117.4  735.61   136.9  732.37   234.8  717.48   244.5  714.38   254.3  710.57
   264.1  708.49   410.8  700.92   537.1  693.23   584.9  692.25   594.4  693.22
     604  696.75   652.1  725.26   661.9  730.63   671.6  733.64   681.4  734.42
   720.4  734.26   808.2  731.78   895.9  724.88   915.4  722.64   954.4  716.19
   964.2  714.95   973.9  714.75   993.4   716.5  1110.4  733.42  1139.7  736.82
#Mann= 3 , 0 , 0
       0     .08       0   537.1    .045       0   594.4     .08       0
Bank Sta=537.1,594.4
XS Rating Curve= 0 ,0
Exp/Cntr=0.3,0.1

Type RM Length L Ch R = 1 ,52735.2 ,265.5,259,250.4
XS GIS Cut Line= 4
     1871185.543      665540.397     1871519.744      665783.453
     1871666.253       665870.68     1872172.956      666111.144
#Sta/Elev= 30
       0  829.43    19.7  822.85    29.5  818.59   108.2  778.75   177.1  748.94
     246  721.09   255.8  718.73   285.3  715.94   314.8   708.7   324.7  707.24
   441.7  693.89     489  692.22     508  692.75   517.4  695.38   526.9   699.5
   536.4  701.18   593.6  703.23     692  716.23     751  721.36   780.5  722.85
   859.3  722.67   928.1  719.01   967.5  715.41  1006.9  709.44  1016.7  709.28
  1026.5  710.94  1056.1  721.05  1075.7  726.22  1115.1  734.17  1144.6  738.14
#Mann= 3 , 0 , 0
       0      .1       0   441.7    .045       0   517.4     .07       0
Bank Sta=441.7,517.4
XS Rating Curve= 0 ,0
Exp/Cntr=0.3,0.1

Type RM Length L Ch R = 1 ,52476.2 ,181.8,174,166.1
XS GIS Cut Line= 4
     1870714.623      665794.304     1871209.414      665976.595
     1871539.276       666043.87     1872110.022      666126.335
#Sta/Elev= 30
       0  755.92     9.8  753.17    29.3  756.37    48.8  764.05    78.1  780.34
   117.2  796.68   136.7  802.37     166  807.44   224.6  809.96     293  805.33
   351.5  810.77   400.4  809.24   478.5  798.16   517.5   780.8   527.3  779.29
   565.8  781.41     585  778.19   642.7  749.62   700.4  710.72   729.3  696.38
   742.7  693.45   767.8  692.24     787  693.18   796.6  695.63   815.9  698.88
  1030.1  702.27  1147.4  707.59  1303.8  705.74  1333.1  709.27  1440.6  733.51
#Mann= 3 , 0 , 0
       0      .1       0   729.3    .045       0   796.6     .05       0
Bank Sta=729.3,796.6
XS Rating Curve= 0 ,0
Exp/Cntr=0.3,0.1

Type RM Length L Ch R = 1 ,52302.2 ,367.4,361.5,355.5
XS GIS Cut Line= 4
     1870593.095      666312.967     1871354.814       666204.46
     1871519.744      666178.418     1872136.064      666182.759
#Sta/Elev= 30
       0  792.73    48.7  785.44   146.1  796.21   175.3  796.29     224  793.62
   292.2   798.4   311.7  797.95   340.9  793.12     409  777.29   477.2  757.32
   516.2  748.74   633.1  732.56   681.8  723.84     711  715.68   749.9  702.45
   759.7  700.46   838.2  694.83   857.8  690.54   867.6  690.24   897.1   691.1
   906.9  692.64   916.7  696.45   926.6  699.17  1171.2  702.22  1259.2  705.16
  1308.1  703.29  1376.6  711.41  1435.3  727.45  1474.4  734.14  1552.7  737.57
#Mann= 3 , 0 , 0
       0      .1       0   838.2    .045       0   916.7     .05       0
Bank Sta=838.2,916.7
XS Rating Curve= 0 ,0
Exp/Cntr=0.3,0.1

Type RM Length L Ch R = 1 ,51940.7 ,410.3,413.4,416.7
XS GIS Cut Line= 5
     1871033.633      666740.484     1871500.213      666560.363
     1871690.289      666478.102     1872170.786      666250.033
     1872404.701      666157.116
#Sta/Elev= 30
       0  788.33    88.3  744.37   137.3  718.67   147.1   714.1   156.9  710.37
   166.7   707.6   176.5  705.83   196.1  704.35   284.4  702.82   411.9  701.89
     519  698.01   528.4  697.45   537.8  695.77   556.6  690.56     566  690.16
   594.3  691.64   613.1  696.88   622.5  698.57   631.9  698.88     920  701.21
  1084.4  698.62  1094.1  700.41  1113.4  706.96  1190.8   730.8  1200.4  733.49
  1210.1  735.16  1219.8  735.89  1355.3  740.08  1452.1  741.52  1490.8  741.19
#Mann= 3 , 0 , 0
       0     .05       0   537.8    .045       0   613.1     .05       0
Bank Sta=537.8,613.1
XS Rating Curve= 0 ,0
Exp/Cntr=0.3,0.1

Type RM Length L Ch R = 1 ,51527.4 ,391.1,387.5,384
XS GIS Cut Line= 5
     1871261.859      666927.159     1871708.546      666907.585
     1871890.838      666853.331     1872615.664      666736.144
      1873168.59      666591.144
#Sta/Elev= 30
       0  740.33   126.4  707.79   155.5  702.97   349.9  701.06   466.1  697.18
   485.2  694.53   494.7  691.41   511.8     690   580.2  691.54   599.3  694.94
   608.8  696.92   656.9  700.28   666.7  704.76   686.3  721.27     696  726.28
   705.8  728.02   754.8  727.86     794  724.55   882.1  705.52   921.2   703.2
  1077.8  710.66    1166  724.66  1224.7  727.85  1332.4  729.49  1458.8  726.93
    1575  727.41  1633.1  724.23  1681.6  728.22  1826.9  745.47  1943.2  752.16
#Mann= 3 , 0 , 0
       0     .05       0   485.2    .045       0   599.3     .06       0
#XS Ineff= 2 , 0
                          678.93          713.24
Permanent Ineff=
       F       F
Bank Sta=485.2,599.3
XS Rating Curve= 0 ,0
Exp/Cntr=0.3,0.1

Type RM Length L Ch R = 1 ,51139.9 ,402,402,401.4
XS GIS Cut Line= 4
      1871448.13      667207.064     1871929.901      667228.766
     1872114.362       667144.13     1872674.258      666924.946
#Sta/Elev= 30
       0  815.12    88.6   791.9   108.3  785.83   255.9  730.87   314.9  707.87
   334.6  702.57   354.3  700.84   423.2  698.62   530.6  696.97   540.2  696.36
   549.9  694.08   559.6  690.97   578.9   689.3   607.9  689.72   617.6  691.24
   627.2  694.17   636.9  696.33   685.2  699.84   704.6  702.72   772.5  728.17
   811.3  738.99   830.7  743.39   850.1   743.1   927.7  734.18   985.8  731.37
  1024.6  731.58  1121.6  733.84  1179.8  736.87  1228.3  740.22  1286.5  748.46
#Mann= 3 , 0 , 0
       0     .06       0   549.9    .045       0   627.2     .07       0
Bank Sta=549.9,627.2
XS Rating Curve= 0 ,0
Exp/Cntr=0.3,0.1

Type RM Length L Ch R = 1 ,50737.9 ,385.6,390.2,394.8
XS GIS Cut Line= 4
     1871658.633       667450.12     1872212.019      667515.224
       1872387.8      667432.759     1872774.085      667237.446
#Sta/Elev= 30
       0  814.31    78.2  814.22    97.8  811.68   127.1  805.66   205.3  783.76
     303  752.17   439.9  700.22   449.7  698.44   469.2   697.4   557.2  698.06
   586.3  697.18   615.4  695.61   625.2  693.35   634.9  690.62   654.3  689.32
     664  689.67   673.7  691.57   683.4  695.85   693.1  698.62   741.7  700.29
   761.2  704.45   790.7  714.82   849.7   739.8   898.9  754.54   908.8  755.45
     958  753.01  1026.8  755.37  1095.7  753.26  1154.7  748.59  1184.2  748.14
#Mann= 3 , 0 , 0
       0     .06       0   625.2    .045       0   673.7     .08       0
Bank Sta=625.2,673.7
XS Rating Curve= 0 ,0
Exp/Cntr=0.3,0.1

Type RM Length L Ch R = 1 ,50347.7 ,388.8,409.4,428.2
XS GIS Cut Line= 4
     1871751.949      667569.477     1872413.841      667827.724
     1872576.602      667788.661     1872902.123      667699.686
#Sta/Elev= 30
       0  805.82    68.1  799.68   116.8  791.97   155.7  787.38     399  746.41
   603.4  721.58   622.9  717.57   681.3  700.07   710.5  697.54   747.7  696.46
   766.3  692.65   775.6  690.13   784.9   689.3   812.8  689.78   822.1  692.08
   840.7  697.87   897.2  699.68   906.8  701.07   916.4  704.52   926.1  709.94
   945.4  717.36     955  724.38   983.9   749.4   993.6  755.72  1012.8  765.59
  1041.8  776.06  1070.7  783.09  1109.3  787.14  1128.6  790.45  1215.3   811.1
#Mann= 3 , 0 , 0
       0     .06       0   766.3    .045       0   822.1      .1       0
Bank Sta=766.3,822.1
XS Rating Curve= 0 ,0
Exp/Cntr=0.3,0.1

Type RM Length L Ch R = 1 ,49938.3 ,117.8,121.6,127.2
XS GIS Cut Line= 3
     1871795.352      667628.071     1872500.404      668196.352
     1872952.036      668502.637
#Sta/Elev= 30
       0  790.74   360.3  744.77   438.2     740   584.2  737.56   642.7  728.18
   691.3   714.7   710.8  710.63   847.1   699.6   876.4  695.48   895.8  689.82
   905.6  689.32     925  691.49   934.8  695.85   954.3  703.55     964  710.49
  1012.8  753.24  1051.7   780.1  1110.2  816.92  1119.9  822.14  1129.7  825.18
  1168.7  826.72  1197.9  824.35  1227.1  820.49  1256.4  812.56  1266.1  813.52
  1295.3  823.24  1334.3  830.53  1402.5   829.6  1431.8  836.68  1451.3   839.3
#Mann= 3 , 0 , 0
       0     .05       0   876.4    .045       0   934.8     .07       0
Bank Sta=876.4,934.8
XS Rating Curve= 0 ,0
Exp/Cntr=0.3,0.1

Type RM Length L Ch R = 1 ,49816.7 ,132.7,144.8,156.9
XS GIS Cut Line= 4
     1871787.105      667648.904      1872331.81      668187.099
     1872495.005      668370.693     1873019.744      668814.269
#Sta/Elev= 30
       0  786.42   206.2  758.81   382.9  740.56   579.2  737.49   638.1  729.33
   716.6  710.85     864  695.87   883.6  689.79   903.3  689.31     923   692.3
   932.8  697.04   952.4  705.72  1001.6  751.06    1031  766.39  1060.5  777.15
  1129.2  789.58  1168.4  792.05  1227.3  784.88    1247  774.47  1266.6  759.14
  1276.4  756.58  1315.7  768.06  1364.8   788.8  1394.2  795.07  1462.9  791.13
  1502.2  795.24  1580.7  809.26  1610.1  811.69    1669  804.48  1698.5  794.53
#Mann= 3 , 0 , 0
       0     .05       0     864    .045       0   932.8      .1       0
#Block Obstruct= 1 ,-1
   741.7   786.8  739.44
Bank Sta=864,932.8
XS Rating Curve= 0 ,0
Exp/Cntr=0.3,0.1
